HEC-RAS study QUEENSFK.prj: QUEENSFK

--- QUEENSFK.g01 (geometry) --- (continued)

Type RM Length L Ch R = 1 ,8638    ,135.7,123.3,108.4
XS GIS Cut Line= 4
2185760.10478138670466.5687207042185783.04328748670512.790336965
2185731.85079422670633.4583567832185729.28481094670660.368873741
#Sta/Elev= 30
       0 1880.11       8 1879.28    16.3 1878.61    19.9 1878.17    25.2 1877.29
    31.8 1876.39    38.6 1875.86    47.6 1874.33    56.4 1873.19    69.4 1871.28
    87.6 1870.09     109 1869.13   112.9 1868.56   117.2  1866.9   121.5 1865.84
   125.9 1865.75   130.2 1865.84   134.6 1866.37   137.5 1866.91   139.5 1867.31
   147.6  1869.4   151.1 1870.19   154.8 1870.59   156.3 1870.66   163.9 1870.46
   190.4 1871.07   198.5 1873.38   202.5 1873.17   206.5 1872.57   209.7 1872.54
#Mann= 7 ,-1,0
       0     .08       0      20      .1       0    81.6     .05       0
   101.6      .1       0   117.2    .045       0   137.5      .1       0
   181.6     .05       0
Bank Sta=117.2,137.5
XS Rating Curve= 0 ,0
Exp/Cntr(USF)=0,0
Exp/Cntr=0.3,0.1

Type RM Length L Ch R = 1 ,8514    ,92.7,97.2,98.4
XS GIS Cut Line= 3
2185625.80920105 670560.84859594 2185703.6426857670659.576975791
2185720.35860186670674.203402436
#Sta/Elev= 29
       0 1874.03    15.7 1871.77      19 1870.81    20.8  1870.1    24.7 1868.05
    25.9 1867.54    27.31867.145    30.4 1866.56    36.1 1866.06    39.31867.109
    41.8 1867.98    44.6 1868.49    46.3 1868.61    51.4 1868.68    58.9 1869.07
    61.5    1869    67.4 1868.56    71.7 1868.48    78.8 1868.48    87.8  1868.6
    93.1 1868.92   102.3 1869.83   112.5 1870.63   122.7 1871.61   125.7 1871.73
   134.2  1871.8   141.4 1872.03   142.4 1872.13   147.9 1873.17
#Mann= 5 ,-1,0
       0     .08       0    27.3    .045       0    39.3     .08       0
      70      .1       0      90     .05       0
Bank Sta=27.3,39.3
XS Rating Curve= 0 ,0
Exp/Cntr(USF)=0,0
Exp/Cntr=0.3,0.1

Type RM Length L Ch R = 1 ,8417    ,81.3,67.5,56.1
XS GIS Cut Line= 4
  2185555.485108670601.7573819752185559.29320265670619.528490348
2185592.71981126670678.765518258 2185613.0296494 670719.38519454
#Sta/Elev= 30
       0 1873.45     3.3 1873.74     7.6 1873.79    13.6 1873.48    20.1  1873.4
      23 1872.89    24.7 1872.52    28.8 1870.48    29.3  1870.3    33.8 1868.02
    37.6 1866.69    38.4  1866.5      43 1866.05    47.6 1866.08    55.3 1866.27
    56.8 1866.36    58.31866.601    70.6 1869.31    75.2 1869.69    88.9 1869.88
    93.5 1869.84   102.3 1869.42   106.8 1869.34   111.3 1869.64   114.4  1870.2
   115.7 1870.36   120.4 1870.64   124.7 1871.08   129.1 1871.21   131.6 1871.06
#Mann= 3 ,-1,0
       0     .08       0    37.6    .045       0    58.3      .1       0
Bank Sta=37.6,58.3
XS Rating Curve= 0 ,0
Exp/Cntr(USF)=0,0
Exp/Cntr=0.3,0.1

Type RM Length L Ch R = 1 ,8350    ,50.3,63.7,76
XS GIS Cut Line= 4
2185504.04163809670679.373829427  2185528.748937670702.970687934
2185590.37837922670711.0213808372185606.20215492 670721.38549124
#Sta/Elev= 19
       0 1870.09     2.6 1870.13     5.7 1869.91    11.2 1869.36    14.2  1869.2
      20 1869.04    27.8 1869.31    31.6 1869.26    33.4 1869.01    37.6 1868.21
    41.7 1867.31    43.8 1867.07    45.7 1866.85    49.7 1866.74    57.11867.091
    92.7 1869.21    98.5 1869.37     105    1870   115.2 1870.68
#Mann= 4 ,-1,0
       0     .08       0    43.8    .045       0    57.1     .08       0
   74.17      .1       0
#XS Ineff= 2 , 0
           27.93 1870.45
Permanent Ineff=
       F       F
Bank Sta=43.8,57.1
XS Rating Curve= 0 ,0
Exp/Cntr(USF)=0,0
Exp/Cntr=0.3,0.1

Type RM Length L Ch R = 1 ,8286    ,43.8,42.4,41.6
XS GIS Cut Line= 3
2185511.33550675670696.1869470782185538.17114976670796.126583108
2185562.77308668670819.041252018
#Sta/Elev= 23
       0 1868.85       8  1868.6    24.3  1867.5    34.2 1867.34    42.4 1866.55
    54.9 1865.52    55.51865.409      59 1864.82    63.2  1864.9    67.21865.398
    75.6 1866.85    79.7 1867.43    83.9 1867.63    86.4 1867.58    92.1  1867.7
    96.3 1868.34   100.4 1869.33   105.6 1869.84   111.7 1870.27   122.6 1870.41
   128.1 1870.64   131.1 1870.98   137.1 1871.85
#Mann= 4 ,-1,0
       0     .08       0      40      .1       0    55.5    .045       0
    67.2      .1       0
#XS Ineff= 2 , 0
                           84.72         1869.17
Permanent Ineff=
       F       F
Bank Sta=55.5,67.2
XS Rating Curve= 0 ,0
Exp/Cntr(USF)=0,0
Exp/Cntr=0.3,0.1

Type RM Length L Ch R = 1 ,8244    ,56.7,48.7,44
XS GIS Cut Line= 4
2185452.66298908670711.6964582012185472.09569609670724.034684871
2185499.54825043 670804.233158232185505.10045243670838.163281573
#Sta/Elev= 30
       0 1874.85     4.2 1874.29     8.9 1873.43    12.3 1872.44    15.2  1871.1
    18.4 1869.31      23 1867.61    24.2  1867.3    30.3 1866.68    36.9 1866.46
    41.1 1865.92    45.4 1864.79      48 1864.33    52.3 1863.74    55.5 1863.48
    58.1  1863.2    66.5 1862.92    70.7 1863.11    72.7 1863.46    79.2 1864.31
    83.4 1864.53    91.9  1866.1    97.4 1866.54   108.7 1868.73   112.6 1869.34
   120.9 1869.25     125 1869.57   133.1 1871.15     137 1870.85   142.2 1870.71
#Mann= 4 ,-1,0
       0     .08       0   33.02      .1       0    55.5    .045       0
    72.7      .1       0
Bank Sta=55.5,72.7
XS Rating Curve= 0 ,0
Exp/Cntr(USF)=0,0
Exp/Cntr=0.3,0.1

Type RM Length L Ch R = 1 ,8195    ,56.4,46.7,40.9
XS GIS Cut Line= 4
2185398.37479173670748.7111382122185421.81742241670763.825465884
2185465.92658276670815.3375622332185480.42399909670830.760345571
#Sta/Elev= 30
       0 1883.52     2.1 1882.88     4.5  1881.9     7.4  1880.6    10.3    1879
    11.7 1878.08    13.2  1876.7    15.6 1874.66      23 1869.91    25.9 1868.27
    29.7 1866.27    31.5  1865.4    34.9 1863.95    37.7 1862.97    40.2 1862.43
    43.8 1861.91    50.7 1861.41    56.1 1861.25    61.7 1861.39    67.4 1861.38
    70.2 1861.62    73.1 1862.01    75.9 1862.46    82.3 1863.85    87.3 1865.28
    92.9 1867.41    98.6 1868.65   109.2 1870.25   114.7 1870.67   116.9 1870.59
#Mann= 3 ,-1,0
       0      .1       0    43.8    .045       0    73.1      .1       0
Bank Sta=43.8,73.1
XS Rating Curve= 0 ,0
Exp/Cntr(USF)=0,0
Exp/Cntr=0.3,0.1

Type RM Length L Ch R = 1 ,8148    ,52.5,51.8,50.8
XS GIS Cut Line= 2
2185373.28646228670808.2953265522185450.03005887670839.895631031
#Sta/Elev= 20
       0 1874.56     3.1  1873.2       9 1870.24    16.1 1867.07    21.3  1864.4
    24.3 1863.01    29.1  1861.6    30.5 1861.32    33.4 1860.79    37.7 1860.59
    42.1 1860.52    46.4 1860.77    50.7 1861.33    51.9 1861.49      58 1862.67
    63.7 1863.93    72.3 1866.98    76.4 1867.94      81 1868.47      83 1868.55
#Mann= 3 ,-1,0
       0      .1       0    30.5    .045       0    50.7      .1       0
Bank Sta=30.5,50.7
XS Rating Curve= 0 ,0
Exp/Cntr(USF)=0,0
Exp/Cntr=0.3,0.1

Type RM Length L Ch R = 1 ,8097    ,39,37.8,37.7
XS GIS Cut Line= 2
2185347.49029536670856.018235357 2185432.6176462670885.683827317
#Sta/Elev= 19
       0 1867.02     3.5 1866.48    10.9 1865.54    30.4 1863.32    34.6 1862.65
    41.61860.568    43.1 1860.11    47.3 1859.85    55.8 1860.08    58.9 1860.63
      60 1860.85    61.1 1861.18    64.3 1862.28    68.5 1864.42    72.7 1866.07
    76.8 1867.17    81.2 1867.88    86.3 1868.27    90.1 1868.37
#Mann= 3 ,-1,0
       0      .1       0    41.6    .045       0    58.9      .1       0
Bank Sta=41.6,58.9
XS Rating Curve= 0 ,0
Exp/Cntr(USF)=0,0
Exp/Cntr=0.3,0.1

Type RM Length L Ch R = 1 ,8059    ,49.5,71.9,85.3
XS GIS Cut Line= 3
2185347.57728004670897.1725823412185411.55327018670917.355483993
2185434.02102862670922.686816505
#Sta/Elev= 18
       0  1865.6     4.8 1864.85       9 1863.98    13.3 1862.79    21.6  1860.7
    25.8 1860.39    35.6 1859.95    38.4 1859.97    41.71860.693    42.6 1860.89
    46.8 1862.66      51 1864.17    55.2 1865.35    59.3 1866.27    64.3 1866.97
    71.8 1867.59    80.1 1868.04    90.2 1868.27
#Mann= 3 ,-1,0
       0      .1       0    21.6    .045       0    41.7      .1       0
Bank Sta=21.6,41.7
XS Rating Curve= 0 ,0
Exp/Cntr(USF)=0,0
Exp/Cntr=0.3,0.1

Type RM Length L Ch R = 1 ,7987    ,67.1,58.9,49.2
XS GIS Cut Line= 4
2185341.44105585670893.7920767622185341.74951151 670930.18984544
2185338.35649918670973.6820944542185338.04804351670993.423257126
#Sta/Elev= 22
       0 1866.02     3.4 1865.75     8.7 1865.06    15.4 1864.33    19.4  1863.6
    23.4 1862.58    27.4 1862.12    31.4 1863.55    35.4  1865.4    39.4 1865.52
    43.4 1863.51    47.4    1862    51.4 1861.36    55.3 1860.88    59.5 1860.58
    67.5 1860.36    70.4 1860.84    71.5 1860.99    83.5  1864.3    87.5 1864.96
    91.5  1865.3    99.8 1865.32
#Mann= 3 ,-1,0
       0      .1       0    55.3    .045       0    70.4      .1       0
Bank Sta=55.3,70.4
XS Rating Curve= 0 ,0
Exp/Cntr(USF)=0,0
Exp/Cntr=0.3,0.1

Type RM Length L Ch R = 1 ,7928    ,42.3,41.5,41.4
XS GIS Cut Line= 3
2185265.56096182670913.224783768 2185300.1079965670973.682094454
2185307.81938817670988.796422125
#Sta/Elev= 24
       0 1870.73     4.6 1868.78     9.2 1865.58    13.3  1863.3    18.4    1861
      23 1858.63    25.3 1857.79    26.51857.482    27.6  1857.2    28.3 1857.13
    32.2 1856.92    41.4 1857.01      46 1857.45    48.8 1858.28    55.2 1860.49
    59.8  1861.6    64.4    1862    66.4 1862.29    69.6 1862.98    73.6 1863.45
    78.2 1863.78    81.2 1864.11    82.5 1864.33    86.6 1864.72
#Mann= 4 ,-1,0
       0     .05       0      20      .1       0    26.5    .045       0
      46      .1       0
Bank Sta=26.5,46
XS Rating Curve= 0 ,0
Exp/Cntr(USF)=0,0
Exp/Cntr=0.3,0.1

Type RM Length L Ch R = 1 ,7886    ,36.9,37.2,37.1
XS GIS Cut Line= 3
2185224.53635814670929.5729341072185259.39184849670983.244220123
2185269.57088549670991.880978793
#Sta/Elev= 23
       0 1874.42     5.2 1871.26     9.1 1868.81      11 1867.51    13.9 1865.39
    18.6 1861.49    19.7 1860.67    22.6  1858.8    23.4 1858.39    25.5 1857.82
    28.1 1857.25   32.321856.842    37.7  1856.3    42.5 1856.02    45.7 1856.48
    47.2 1856.84      52  1858.8    61.5 1861.82      65 1862.53      67 1862.84
    70.3 1863.07    73.2 1863.14    77.3 1863.05
#Mann= 3 ,-1,0
       0      .1       0   32.32    .045       0    47.2      .1       0
Bank Sta=32.32,47.2
XS Rating Curve= 0 ,0
Exp/Cntr(USF)=0,0
Exp/Cntr=0.3,0.1

Type RM Length L Ch R = 1 ,7849    ,41.7,41,40.5
XS GIS Cut Line= 4
2185192.76542447670949.005641113 2185204.4867398670965.970702785
2185226.38709214671000.2092817952185247.67053315671001.443104462
#Sta/Elev= 22
       0 1873.72     9.9 1868.72    14.8 1865.84    19.7 1862.78    24.4 1859.28
    25.6 1858.47    28.5  1856.7    29.2 1856.38   30.541856.167    33.9 1855.76
    38.7  1855.7    43.4 1855.83    45.4 1856.16    48.2 1856.77    52.9  1858.5
    54.6 1859.01    57.7 1859.79    61.3 1860.41    67.1 1861.18    71.4  1861.6
    75.2 1861.85    82.6  1862.1
#Mann= 3 ,-1,0
       0      .1       0   30.54    .045       0    45.4      .1       0
Bank Sta=30.54,45.4
XS Rating Curve= 0 ,0
Exp/Cntr(USF)=0,0
Exp/Cntr=0.3,0.1

Type RM Length L Ch R = 1 ,7808    ,37.8,37.6,37.7
XS GIS Cut Line= 4
2185158.71068428670967.2655837832185166.70585516670984.005472818
2185191.94061326671019.9837417892185206.93155867671028.478610852
#Sta/Elev= 20
       0 1872.74     3.4 1871.09     6.6 1869.32      11  1866.4      20 1859.79
    23.3 1857.64    24.9 1856.74    26.2 1856.21    28.1 1855.64    29.8 1855.34
    34.6 1855.15    39.5 1855.19    44.4  1855.6    46.3 1856.04      52 1857.81
    54.2 1858.37    63.5 1859.82    66.5 1860.22    72.3 1860.66    79.7 1860.87
#Mann= 3 ,-1,0
       0      .1       0    28.1    .045       0    44.4      .1       0
Bank Sta=28.1,44.4
XS Rating Curve= 0 ,0
Exp/Cntr(USF)=0,0
Exp/Cntr=0.3,0.1

Type RM Length L Ch R = 1 ,7771    ,50.3,47.2,44.8
XS GIS Cut Line= 4
2185126.22292802670989.1411365292185134.44841247671003.193005792
2185159.46759433671039.1795002482185179.00311989 671046.03407062
#Sta/Elev= 20
       0 1866.01     9.3 1861.25    13.9 1859.34    18.7 1858.29    23.6 1857.35
    30.4 1855.75      331855.248    38.2  1854.5    41.9 1854.29    43.1 1854.32
    44.8 1854.61    47.11855.291    47.7 1855.48    50.6 1857.06    52.8 1858.09
    54.3 1858.46    56.3 1858.79    65.1 1859.56    73.6 1859.87    80.8 1860.04
#Mann= 3 ,-1,0
       0      .1       0      33    .045       0    47.1      .1       0
Bank Sta=33,47.1
XS Rating Curve= 0 ,0
Exp/Cntr(USF)=0,0
Exp/Cntr=0.3,0.1

Type RM Length L Ch R = 1 ,7724    ,56.3,59.7,62.3
XS GIS Cut Line= 3
2185076.66815926671020.431789321 2185128.7121195671067.821411649
2185152.83005229671064.013316998
#Sta/Elev= 20
       0 1859.12       3 1858.68    14.3 1856.75    22.8 1855.91    30.8 1854.86
    36.8 1853.66    39.8 1853.28    42.7 1853.03    48.3 1853.17    51.1 1853.73
    56.8 1855.59    59.6 1856.31    65.3 1856.81    66.5 1857.03    70.4 1858.07
    73.9 1858.39    77.9 1858.64    85.8 1858.67    90.1 1858.53    94.8 1858.65
#Mann= 3 ,-1,0
       0      .1       0    36.8    .045       0    51.1      .1       0
Bank Sta=36.8,51.1
XS Rating Curve= 0 ,0
Exp/Cntr(USF)=0,0
Exp/Cntr=0.3,0.1

Type RM Length L Ch R = 1 ,7664    ,42.8,52.2,63.8
XS GIS Cut Line= 3
2185044.93403717671058.5127358352185083.43810531671116.480398861
2185082.59186205671138.059601886
#Sta/Elev= 27
       0 1857.44     4.3 1856.64       8 1855.61    12.8 1854.48    15.8 1854.39
    22.4 1854.45    24.5 1854.38    27.3 1854.11      32 1852.99    34.8 1852.63
    36.8 1852.55    41.6 1852.61    44.7 1852.83    46.4 1853.03    53.3 1854.53
      56 1855.27    56.5 1855.48    60.8 1857.77    63.7 1859.05    65.6 1859.79
    67.7 1860.36    70.3 1860.93    74.3 1861.54    78.3 1862.36    82.3 1864.08
    86.3 1865.58    91.2  1866.8
#Mann= 4 ,-1,0
       0      .1       0      32    .045       0    46.4      .1       0
   79.59     .06       0
Bank Sta=32,46.4
XS Rating Curve= 0 ,0
Exp/Cntr(USF)=0,0
Exp/Cntr=0.3,0.1

Type RM Length L Ch R = 1 ,7612    ,57.9,69.1,85.5
XS GIS Cut Line= 4
2185041.32072791671053.7897415922185030.54790182671073.321992812
2185011.08430693671126.6353179322185013.19991507671147.791399328
#Sta/Elev= 24
       0 1857.71     9.2  1856.4    12.2 1856.22    22.3 1856.29    26.4 1856.09
    34.9 1853.96    39.6 1853.87    43.4 1854.02    47.7 1853.82    52.1 1852.35
      531852.167    56.2 1851.55    60.5  1851.5    64.6 1851.98      65 1852.22
    67.7 1853.91      69 1854.82    70.8 1856.24    73.3 1857.94      74 1858.21
    77.1 1858.86    82.4 1858.93    89.7 1858.78   100.3 1858.21
#Mann= 4 ,-1,0
       0      .1       0      53    .045       0      65      .1       0
   79.06     .06       0
Bank Sta=53,65
XS Rating Curve= 0 ,0
Exp/Cntr(USF)=0,0
Exp/Cntr=0.3,0.1

Type RM Length L Ch R = 1 ,7542    ,57.1,45.4,36.1
XS GIS Cut Line= 2
2185041.64857989 671051.494777762184973.72833134671048.066965936
#Sta/Elev= 28
       0 1857.89     1.5 1857.66     5.5 1856.83     7.4 1856.15     9.5 1855.43
    11.2 1854.42    11.8 1854.08    13.5 1853.08      15 1852.28      16 1851.85
    17.5 1851.08    18.9 1850.83    20.2 1850.63    21.5 1850.39    25.5 1850.53
    29.5 1850.74    33.5 1851.19    37.1 1851.79    37.9 1851.92    41.7  1852.4
    45.5 1852.81    49.5 1853.28    53.9 1853.98      57 1854.64    57.5 1854.74
    58.2 1854.88    65.6 1856.57      68 1856.92
#Mann= 4 ,-1,0
       0      .1       0    17.5    .045       0    33.5      .1       0
   68.01     .06       0
Bank Sta=17.5,33.5
XS Rating Curve= 0 ,0
Exp/Cntr(USF)=0,0
Exp/Cntr=0.3,0.1

Type RM Length L Ch R = 1 ,7497    ,61.7,53.3,45.5
XS GIS Cut Line= 4
2185036.44765025670962.7275647992185027.53670876670985.690375547
2184981.95381579671032.9869111172184970.98650319671044.296952231
#Sta/Elev= 23
       0 1871.88     5.2 1869.62     8.3 1868.12    19.8 1862.34    29.5 1857.13
      35 1854.47      41  1852.2    43.6 1851.46    46.4 1850.77    51.7 1850.15
    54.9 1850.09    57.8 1850.16    60.71850.717    62.8 1851.29    66.3 1852.03
    68.4 1852.58    73.9 1853.41    80.4  1853.9    86.1  1854.5    88.9 1854.94
    90.6 1855.31    98.6 1856.54   106.1 1857.05
#Mann= 4 ,-1,0
       0      .1       0    46.4    .045       0    60.7      .1       0
  100.32     .06       0
Bank Sta=46.4,60.7
XS Rating Curve= 0 ,0
Exp/Cntr(USF)=0,0
Exp/Cntr=0.3,0.1

Type RM Length L Ch R = 1 ,7444    ,42.2,40.7,38.9
XS GIS Cut Line= 2
2184961.04737615670952.1029807222184953.50734874671028.531440375
#Sta/Elev= 19
       0 1870.97     1.1 1870.24     5.1 1867.32    13.1 1860.53    17.2 1857.46
    21.2 1854.17    25.2 1851.64    29.2 1850.05    33.2 1849.58    41.3 1849.76
   43.671850.062    45.3 1850.27    49.3 1852.25    53.3 1853.67    53.7 1853.75
    57.4 1854.32    61.4 1854.77    69.4 1855.85    76.8 1856.66
#Mann= 4 ,-1,0
       0      .1       0    29.2    .045       0   43.67      .1       0
    76.8     .06       0
Bank Sta=29.2,43.67
XS Rating Curve= 0 ,0
Exp/Cntr(USF)=0,0
Exp/Cntr=0.3,0.1

Type RM Length L Ch R = 1 ,7403    ,37.5,36.3,35.3
XS GIS Cut Line= 4
2184918.54903984670954.8448088712184916.49266873670965.469392948
2184918.20631132671017.9068562972184927.80270984671034.357825191
#Sta/Elev= 18
       0 1865.76     2.4 1864.29     6.5 1861.51    14.1 1855.99    18.5 1852.96
    22.5 1850.44    25.7 1849.64    26.5 1849.41    30.5 1849.38    34.5 1849.14
    38.5  1849.1    42.5 1849.69    50.6 1853.49    58.6 1854.89    62.6 1855.48
    67.1 1855.93    71.7 1856.18    82.3 1856.42
#Mann= 4 ,-1,0
       0      .1       0    25.7    .045       0    42.5      .1       0
   73.29     .06       0
Bank Sta=25.7,42.5
XS Rating Curve= 0 ,0
Exp/Cntr(USF)=0,0
Exp/Cntr=0.3,0.1

Type RM Length L Ch R = 1 ,7367    ,60.5,59,53.1
XS GIS Cut Line= 4
2184877.06459085670951.6532913642184877.68150219670963.991518034
2184885.39289385671024.4488287192184888.78590619671050.667560394
#Sta/Elev= 24
       0 1865.17     1.5 1864.17     5.5 1860.95     9.5  1858.1    13.6 1855.41
    17.6 1853.24    21.6  1851.7    25.6 1850.33    29.7 1849.42    33.7 1848.99
    37.7 1848.59    41.8  1848.3    45.8  1848.4    49.8 1848.93    57.9  1851.6
    61.9 1852.44      66 1853.11      70 1853.55    73.3 1853.81    82.1 1854.22
    86.1 1854.49    90.2 1854.84    98.2 1855.88    99.7 1855.96
#Mann= 4 ,-1,0
       0      .1       0    33.7    .045       0    49.8      .1       0
    73.3     .06       0
Bank Sta=33.7,49.8
XS Rating Curve= 0 ,0
Exp/Cntr(USF)=0,0
Exp/Cntr=0.3,0.1

Type RM Length L Ch R = 1 ,7308    ,16.6,16.8,17.6
XS GIS Cut Line= 3
2184812.01104857670955.7288814552184835.08409105671024.926574423
2184832.03880562671095.406032184
#Sta/Elev= 27
       0 1853.87       2 1853.31     4.4 1853.02     5.7 1852.66     7.6 1852.43
      10 1851.96    14.2 1851.52    17.1 1851.37    26.6 1850.47    35.3 1849.48
    39.5 1848.89    47.9 1848.08    60.6 1847.95    64.8 1848.23      69 1848.92
    72.9 1849.69    81.2  1850.7    85.2 1851.06    97.2  1851.8   105.2 1852.18
   110.5 1852.62   116.2 1853.19   124.6 1854.23   129.2 1854.88   137.3 1855.79
   141.3 1856.09   143.5 1856.12
#Mann= 4 ,-1,0
       0      .1       0    39.5    .045       0      69      .1       0
   72.94     .06       0
#XS Ineff= 2 , 0
           32.21    1855   78.33         1855.55
Permanent Ineff=
       F       F
Bank Sta=39.5,69
XS Rating Curve= 0 ,0
Exp/Cntr(USF)=0,0
Exp/Cntr=0.3,0.1

Type RM Length L Ch R = 1 ,7291    ,42.8,47.9,52.5
XS GIS Cut Line= 4
2184793.67577802670960.1011382772184809.94245394670998.558192903
2184818.21683244671028.7878825432184817.04149459671094.653815956
#Sta/Elev= 30
       0 1854.34     6.4 1854.25     9.9  1854.1    11.9 1853.88    16.7 1853.59
      21 1853.07    24.1 1852.83    27.2 1852.86    31.6  1852.3    33.3 1851.91
    37.2 1851.23    40.3 1850.58      48 1848.51      49 1848.27    52.2 1847.78
    56.9 1847.66    61.1 1847.82    65.2  1848.6    68.5  1849.5    73.1 1850.33
    81.5 1852.32    85.5 1852.94    93.5 1853.94    99.9 1854.61   105.5 1854.93
   109.5 1854.78   121.5 1855.14   124.4 1855.51   129.5 1855.96     139 1855.79
#Mann= 4 ,-1,0
       0      .1       0      48    .045       0    65.2      .1       0
   71.76     .06       0
Bank Sta=48,65.2
XS Rating Curve= 0 ,0
Exp/Cntr(USF)=0,0
Exp/Cntr=0.3,0.1

Type RM Length L Ch R = 1 ,7243    ,35.6,39.3,41.8
XS GIS Cut Line= 3
2184772.79294524670967.1299891422184765.55756541671055.477785054
2184764.79594648671069.948544729
#Sta/Elev= 26
       0 1853.39     2.5 1853.15    14.1 1852.39    18.1 1851.99    22.1 1851.48
    26.1  1850.9    30.1 1850.18    34.2  1849.2    38.2    1848    42.2 1847.26
    46.2 1847.31    50.2 1847.71    54.2 1847.71    58.4 1847.45    62.3 1847.68
    63.31847.993    65.5 1848.62    70.3 1850.23    78.3 1852.25    82.3 1852.69
    86.3  1852.8    91.6 1853.29    94.4 1853.47    98.4 1853.32   102.4 1852.55
   103.1 1852.52
#Mann= 3 ,-1,0
       0      .1       0    38.2    .045       0    63.3     .06       0
Bank Sta=38.2,63.3
XS Rating Curve= 0 ,0
Exp/Cntr(USF)=0,0
Exp/Cntr=0.3,0.1

Type RM Length L Ch R = 1 ,7204    ,48.2,58.9,62.4
XS GIS Cut Line= 3
2184762.51108968670940.0925171182184743.85142589670969.034036468
2184720.62204852671045.957548425
#Sta/Elev= 28
       0 1856.12     2.5 1855.67     6.1 1854.63    10.8 1853.41    15.6 1852.64
    19.1  1852.3    25.1 1851.91    34.4 1851.63    38.8 1851.61    43.9 1851.38
    47.1 1851.09    51.3 1850.55    56.8 1849.47    59.7 1848.98    63.8 1848.69
    66.4 1848.35    69.41847.843    72.2 1847.35    84.7    1847    88.9 1847.25
    90.8 1847.83    93.1 1848.58    97.3 1850.77   101.4 1852.62   105.6  1853.4
   108.1 1853.72   109.8 1853.92   114.8  1854.3
#Mann= 4 ,-1,0
       0      .1       0    69.4    .045       0    90.8      .1       0
   94.44     .06       0
Bank Sta=69.4,90.8
XS Rating Curve= 0 ,0
Exp/Cntr(USF)=0,0
Exp/Cntr=0.3,0.1

Type RM Length L Ch R = 1 ,7145    ,70.9,71.9,72.1
XS GIS Cut Line= 3
2184735.85442713670913.0550450932184723.28771478670935.903613001
2184661.21577196671014.350362819
#Sta/Elev= 27
       0 1858.55     5.7 1856.69     7.6 1856.24     9.3 1855.74    11.6 1854.84
    13.8 1854.08    18.4 1852.82      23 1851.89    29.2 1850.83    37.7 1849.71
    43.4 1848.77    50.4 1848.09    53.2  1847.7    58.3 1846.01    61.21845.568
    63.4 1845.28    69.1 1845.25    78.11845.568    83.8 1845.62    89.1 1845.38
      94 1845.74    95.6    1846   104.2 1848.19   111.8 1850.63   114.6 1851.35
   119.5 1851.86   126.1 1852.04
#Mann= 3 ,-1,0
       0      .1       0    61.2    .045       0    78.1      .1       0
Bank Sta=61.2,78.1
XS Rating Curve= 0 ,0
Exp/Cntr(USF)=0,0
Exp/Cntr=0.3,0.1

Type RM Length L Ch R = 1 ,7073    ,80.3,81.9,83.5
XS GIS Cut Line= 3
 2184682.6164397670872.821577069 2184669.2911549670892.809504275
2184601.83190058670972.761213099
#Sta/Elev= 30
       0 1862.28    11.6 1857.81    14.9 1856.26    22.2 1852.46    25.1 1851.07
    29.7 1849.18      35 1847.64    40.2 1846.92    42.1 1846.76    44.9 1846.29
    47.8  1845.6    50.7 1844.58    53.5  1844.2    56.8 1843.72    66.4 1843.74
    67.7 1843.83    70.5 1844.31    76.2  1845.3    76.8 1845.28    82.1 1844.17
    84.7 1844.12    87.3 1844.31    90.4 1845.05    97.8 1847.07   104.6 1847.68
   110.2 1849.19   113.1 1849.83   115.9 1850.06   121.6 1850.31   128.6 1850.29
#Mann= 3 ,-1,0
       0      .1       0    53.5    .045       0    70.5      .1       0
Bank Sta=53.5,70.5
XS Rating Curve= 0 ,0
Exp/Cntr(USF)=0,0
Exp/Cntr=0.3,0.1

Type RM Length L Ch R = 1 ,6991    ,25.7,25.2,24.9
XS GIS Cut Line= 3
2184634.03467219670835.6218236582184623.20787828670847.003837761
2184549.91881186670904.191518379
#Sta/Elev= 29
       0 1865.39     2.4 1864.27     8.1 1861.24    14.3 1858.25    19.4 1855.47
    22.3 1853.99      28 1851.23    30.8 1849.96    32.2 1849.39    34.8 1848.53
    38.8  1847.7    45.3 1846.94    47.9 1846.54    51.8 1846.08    59.3 1844.71
    64.8 1844.44    70.3 1844.41    75.4 1843.62    79.3 1842.72    80.4 1842.54
    82.1 1842.51      85 1842.66    85.5 1842.79   87.461843.608    90.7  1845.3
    93.5 1846.34    96.4 1847.21   100.7 1847.55   108.7 1847.81
#Mann= 3 ,-1,0
       0      .1       0    75.4    .045       0   87.46      .1       0
Bank Sta=75.4,87.46
XS Rating Curve= 0 ,0
Exp/Cntr(USF)=0,0
Exp/Cntr=0.3,0.1

Type RM Length L Ch R = 1 ,6966    ,176.9,153,120.9
XS GIS Cut Line= 3
2184604.43584666670821.5564783452184588.82265859670840.596951602
2184540.49713786670880.568269715
#Sta/Elev= 25
       0 1862.04      15 1852.89    20.2 1850.23    25.5 1847.66    28.3 1846.66
    31.2 1845.75      34 1845.38    46.2 1844.63    51.4 1844.46    53.9 1844.15
    56.6 1843.73    57.61843.497    61.8 1842.55    65.3 1842.42      67 1842.51
    68.1 1842.69    69.5 1843.03   70.951843.513    73.8 1844.91    76.6 1846.07
    77.4  1846.3    79.5 1846.81    82.3 1847.35    85.2 1847.54    87.3 1847.58
#Mann= 3 ,-1,0
       0      .1       0    57.6    .045       0   70.95      .1       0
Bank Sta=57.6,70.95
XS Rating Curve= 0 ,0
Exp/Cntr(USF)=0,0
Exp/Cntr=0.3,0.1

Type RM Length L Ch R = 1 ,6813    ,37.6,35.8,34.4
XS GIS Cut Line= 3
2184405.47574284670843.8747326622184419.94514798 670853.01327447
 2184516.8443841670883.554581972
#Sta/Elev= 30
       0 1847.51     3.2 1847.58     7.9 1848.23    12.7 1848.15    17.1 1847.89
    21.5 1847.77    25.7 1846.86    29.9 1844.98    34.1 1843.62    38.3    1843
    44.3  1842.3    50.9 1841.09    55.7 1842.42    57.6 1842.87    59.3 1843.13
    63.5 1842.25    66.91841.387    67.7  1841.2    71.9 1840.72    74.8  1840.7
    80.3 1840.73    84.5 1841.37    87.6 1842.41    92.8  1844.6    97.2 1845.66
   101.2 1846.18   105.4 1846.32   109.6 1846.23   113.8  1846.3   118.7 1846.51
#Mann= 3 ,-1,0
       0      .1       0    66.9    .045       0    84.5      .1       0
Bank Sta=66.9,84.5
XS Rating Curve= 0 ,0
Exp/Cntr(USF)=0,0
Exp/Cntr=0.3,0.1

Type RM Length L Ch R = 1 ,6777    ,48.3,47.3,46.2
XS GIS Cut Line= 3
 2184417.4531137670897.6445321822184503.89686229670910.211244531
2184518.36762196670918.208243299
#Sta/Elev= 25
       0 1846.68     2.8 1846.61     6.8 1845.92    14.9 1843.92      23 1842.57
      27 1840.98      31 1839.83    35.1 1839.98    39.1 1840.71    40.81840.436
    43.2 1840.05    47.2 1839.75    51.3 1840.02    52.51840.424    55.3 1841.39
    59.3 1843.36      62 1844.49    63.4 1844.99    67.4 1845.77    71.5 1846.36
    79.5 1847.28    87.7 1847.52    96.8 1848.02   101.4  1848.4   103.9 1848.49
#Mann= 3 ,-1,0
       0      .1       0    40.8    .045       0    52.5      .1       0
Bank Sta=40.8,52.5
XS Rating Curve= 0 ,0
Exp/Cntr(USF)=0,0
Exp/Cntr=0.3,0.1

Type RM Length L Ch R = 1 ,6730    ,65.3,64.5,64.2
XS GIS Cut Line= 3
2184408.53091202670948.4607787152184500.99082331670953.162130136
2184524.49758041670946.371289194
#Sta/Elev= 20
       0 1844.52     3.6 1844.79     7.7 1844.69    11.7 1844.31    15.7 1843.61
    19.7 1842.59    27.7 1839.76    31.7 1839.35    43.7 1839.86    47.7 1839.56
    51.7 1839.39    55.7 1839.85    59.7 1840.94    63.7 1841.75    67.7 1842.41
    83.8 1845.51    87.8 1846.15   100.1 1847.53   104.2 1847.92     117 1848.57
#Mann= 3 ,-1,0
       0      .1       0    43.7    .045       0    55.7      .1       0
Bank Sta=43.7,55.7
XS Rating Curve= 0 ,0
Exp/Cntr(USF)=0,0
Exp/Cntr=0.3,0.1

Type RM Length L Ch R = 1 ,6665    ,56.3,59,62
XS GIS Cut Line= 3
2184404.12013667671014.2796986152184496.28947189671015.324443375
2184510.91589853671028.906125259
#Sta/Elev= 25
       0 1842.47     8.1 1842.68    12.1  1842.5    16.1  1841.7    20.1 1840.74
    24.1 1840.53    28.1 1840.57    32.1 1840.03    37.11838.403    40.1 1837.57
    44.1 1837.46    48.1 1837.84    52.1 1837.75    56.1 1837.54    60.1 1837.81
    61.7 1838.33    64.1 1839.11    68.1 1840.77    76.1 1843.87    80.1 1844.92
    84.1 1845.58    88.1 1846.12    92.2 1846.38    94.9 1846.68   112.1 1848.05
#Mann= 3 ,-1,0
       0      .1       0    37.1    .045       0    61.7      .1       0
Bank Sta=37.1,61.7
XS Rating Curve= 0 ,0
Exp/Cntr(USF)=0,0
Exp/Cntr=0.3,0.1

Type RM Length L Ch R = 1 ,6606    ,68.1,85.6,102.8
XS GIS Cut Line= 4
2184383.06941192671056.4914888812184386.44730199671060.226444639
2184401.96293049671062.9248148122184485.84202428671081.665735655
#Sta/Elev= 29
       0 1841.74     4.1 1842.01     7.4 1842.12    14.9 1842.01      19  1842.1
    23.1 1842.04    35.3 1841.35    39.4 1841.09    43.5 1840.23    47.6  1838.6
    51.7  1838.5    55.8 1839.36    59.9 1838.39    61.4 1837.92      64 1837.11
    68.1 1836.94    72.2 1837.43    74.8 1837.93    76.3 1838.27    78.1  1838.8
    80.4 1839.56    81.5 1840.07    84.5 1841.74    92.7  1847.3    94.9  1848.5
    96.8 1849.63   100.9 1851.24     105 1852.33   106.7 1852.62
#Mann= 3 ,-1,0
       0      .1       0    61.4    .045       0    74.8      .1       0
Bank Sta=61.4,74.8
XS Rating Curve= 0 ,0
Exp/Cntr(USF)=0,0
Exp/Cntr=0.3,0.1

Type RM Length L Ch R = 1 ,6520    ,95.2,93.1,90.1
XS GIS Cut Line= 3
2184378.62065318671028.0066685352184379.14302556671151.808922632
2184381.75488746671166.957721657
#Sta/Elev= 30
       0 1842.04     9.2  1842.5    13.2 1842.43    21.2 1841.77    25.2 1841.55
    42.5  1841.9    45.2  1841.9    49.2 1841.68    53.2 1841.29    57.2 1840.69
    61.2 1839.69    65.2  1838.3    68.91837.282    73.2 1836.78    81.2 1836.99
      88 1836.89    89.2 1836.93    90.3 1837.32    93.2 1838.28     100 1843.12
   101.2 1843.96   105.2 1847.22   110.3 1851.74   113.2 1854.51   116.1 1857.58
   121.2 1862.67   125.2 1865.63   129.3 1866.93   133.3  1867.4   139.2 1867.68
#Mann= 4 ,-1,0
       0      .1       0    68.9    .045       0    90.3      .1       0
     100     .06       0
Bank Sta=68.9,90.3
XS Rating Curve= 0 ,0
Exp/Cntr(USF)=0,0
Exp/Cntr=0.3,0.1

Type RM Length L Ch R = 1 ,6427    ,124,121.8,119.2
XS GIS Cut Line= 4
2184270.78433766670991.8056170052184276.28491883671047.234550264
2184292.78666232671135.2438488732184297.01787859671168.247335851
#Sta/Elev= 30
       0 1841.06    17.5 1840.72    21.5 1840.72    37.6 1841.12    49.1 1840.72
    57.7 1840.14    69.9 1838.52      78 1837.93    82.1 1837.78    86.2 1837.79
    94.3 1837.28    98.4 1836.84   106.5 1836.72   108.7 1836.54   110.6 1836.35
   114.7 1835.35   118.7    1835   122.8 1834.92   126.9 1834.66   130.9    1835
  131.971835.357     135 1836.46   151.2 1846.74   155.3 1848.81   159.3 1850.48
   163.3  1851.9   167.4  1853.2   171.4 1854.75     175 1856.73   178.5 1858.91
#Mann= 4 ,-1,0
       0      .1       0   114.7    .045       0  131.97      .1       0
   135.7     .06       0
Bank Sta=114.7,131.97
XS Rating Curve= 0 ,0
Exp/Cntr(USF)=0,0
Exp/Cntr=0.3,0.1

Type RM Length L Ch R = 1 ,6305    ,101.3,97.4,92.3
XS GIS Cut Line= 4
2184082.91833486671037.502752822 2184157.4723657 671106.09076871
2184185.73689045671178.4022549222184212.81667464671206.328282365
#Sta/Elev= 30
       0 1848.06    17.2 1844.04    29.1  1840.5    31.8 1839.27    37.5 1837.19
    40.3 1836.39    43.1 1836.04      46 1835.82    64.5 1835.76    66.9 1835.93
    72.4 1836.68    82.2 1837.35    91.2 1837.69     100 1837.81   104.6 1837.64
   121.8 1836.53   130.4 1834.23   133.6 1833.98   143.3  1833.5  148.271833.968
   155.2 1835.74   160.5 1836.77   164.7 1837.86   173.7  1839.7   177.6 1840.81
     194 1846.85   202.4 1850.59   211.2  1853.8   216.2 1855.82   217.8 1856.62
#Mann= 3 ,-1,0
       0      .1       0   133.6    .045       0  148.27      .1       0
#XS Ineff= 2 , 0
           99.21 1849.97
Permanent Ineff=
       F       F
Bank Sta=133.6,148.27
XS Rating Curve= 0 ,0
Exp/Cntr(USF)=0,0
Exp/Cntr=0.3,0.1

Type RM Length L Ch R = 1 ,6208    ,65.2,65.2,65.1
XS GIS Cut Line= 3
2184019.10233585671120.0295019282184116.28867244671217.822312846
2184145.61100126671240.670880754
#Sta/Elev= 30
       0 1844.34     7.3 1843.06    12.9 1842.28    35.6 1840.31      44 1839.42
    52.4 1838.09      58 1837.34    66.6    1835    69.3  1834.6    77.9 1834.96
    80.8 1834.82    83.6 1834.46    91.9 1832.96    97.7 1832.57   100.6 1832.71
   103.1 1832.99   109.3  1834.6   114.7 1835.05     120  1836.3   123.2 1836.78
     126    1837   142.8 1837.46   147.9 1838.11   151.6 1839.11   154.4 1840.22
   157.3 1841.63     163 1844.79   168.2 1847.25   173.2 1848.72     175  1849.4
#Mann= 4 ,-1,0
       0      .1       0    91.9    .045       0   103.1      .1       0
  147.87     .06       0
Bank Sta=91.9,103.1
XS Rating Curve= 0 ,0
Exp/Cntr(USF)=0,0
Exp/Cntr=0.3,0.1

Type RM Length L Ch R = 1 ,6143    ,42.9,40.3,36.8
XS GIS Cut Line= 3
2183963.48534854671154.5750321732184068.30667983671261.615401336
2184104.48357902671295.126634268
#Sta/Elev= 30
       0 1845.63     6.7 1844.95    12.4 1843.85    22.1 1841.56    29.6 1840.46
    39.1 1838.39    44.8 1837.55    50.4 1837.02    53.2 1836.96    63.9 1837.45
      82 1837.61    87.2 1836.97    92.8 1834.89    95.7 1834.03     101 1832.89
   104.4 1832.44   112.6 1832.43   115.5 1832.48   118.3 1832.96     124 1834.24
   126.8 1834.68     138 1835.08   143.9 1836.01   149.2 1835.98   160.5 1835.07
   166.4 1835.89   176.9 1838.26   178.6 1838.77   191.9 1844.03   199.1 1847.16
#Mann= 4 ,-1,0
       0      .1       0     101    .045       0   118.3      .1       0
  189.82     .06       0
#XS Ineff= 2 , 0
                          146.54         1839.94
Permanent Ineff=
       F       F
Bank Sta=101,118.3
XS Rating Curve= 0 ,0
Exp/Cntr(USF)=0,0
Exp/Cntr=0.3,0.1

Type RM Length L Ch R = 1 ,6103    ,64.2,69.3,72.6
XS GIS Cut Line= 3
2183949.48080137671221.2094355862184067.37717138671296.784894982
2184092.33496287671324.644755257
#Sta/Elev= 30
       0 1842.73     3.2 1842.89       8 1842.78    14.8 1841.92      27 1840.08
    36.5 1839.52    45.4 1837.96    51.8  1837.1    55.5 1836.32    56.9 1835.83
      65 1833.74    68.5 1832.39    69.7 1832.06    71.4  1831.7    74.5  1831.4
      84 1831.75    85.9  1832.1    88.9 1832.72    93.5 1833.43   103.7  1834.1
   117.7 1835.42     122 1835.94   129.3 1837.56   136.2 1838.86   147.2 1840.54
   152.2 1841.84   163.5 1846.39   167.4 1847.72   172.8 1849.97   177.4 1852.54
#Mann= 4 ,-1,0
       0      .1       0    69.7    .045       0    85.9      .1       0
  170.04     .06       0
Bank Sta=69.7,85.9
XS Rating Curve= 0 ,0
Exp/Cntr(USF)=0,0
Exp/Cntr=0.3,0.1

Type RM Length L Ch R = 1 ,6033    ,63.3,78.1,86.6
XS GIS Cut Line= 4
2183950.71400648671237.0022781422183962.32228159671295.624067471
2183993.08421064671339.7355129062184007.59455454671369.336614448
#Sta/Elev= 27
       0 1840.32     4.3 1839.49    12.4 1838.46    16.5 1837.62    20.6 1836.54
    24.6 1835.71      32 1834.88    36.9 1834.67    45.6 1834.48    57.3 1834.55
      70 1834.29    71.4 1834.16      77 1833.38      84 1831.85      86 1831.51
      91 1831.25    93.8 1831.46    95.8 1831.85    96.7 1832.09    99.6 1833.08
     105  1835.2   122.9 1841.69   125.9 1842.66   128.9 1843.45     133 1844.34
   137.4 1845.43   146.5 1847.18
#Mann= 4 ,-1,0
       0      .1       0      84    .045       0    95.8      .1       0
  123.54     .06       0
#XS Ineff= 2 , 0
            57.2 1838.37
Permanent Ineff=
       F       F
Bank Sta=84,95.8
XS Rating Curve= 0 ,0
Exp/Cntr(USF)=0,0
Exp/Cntr=0.3,0.1

Type RM Length L Ch R = 1 ,5955    ,73.9,68.9,65.2
XS GIS Cut Line= 4
2183940.84697263671224.8135892722183937.94490385671256.155932081
2183903.12007851671376.8819932732183901.95925099671391.392337166
#Sta/Elev= 30
       0 1840.97      12  1839.2    24.5  1837.1    40.2 1835.28    43.4 1835.04
    49.2 1834.81    57.5 1834.32      66 1833.99    75.7 1833.25    86.7 1832.54
    90.8 1832.19      95 1831.38    99.2 1830.26   103.3 1829.76   111.6 1829.74
   115.8 1829.87   118.81830.205     120 1830.35     121 1830.69   124.5 1832.13
   127.4  1833.7   128.3  1834.1   132.5 1835.66   136.6  1836.4   140.8 1836.99
   144.9 1837.42   149.1 1837.41   157.1 1837.03   161.4 1836.94   171.7 1836.94
#Mann= 3 ,-1,0
       0      .1       0    99.2    .045       0   118.8      .1       0
Bank Sta=99.2,118.8
XS Rating Curve= 0 ,0
Exp/Cntr(USF)=0,0
Exp/Cntr=0.3,0.1

Type RM Length L Ch R = 1 ,5886    ,80,68.5,56
XS GIS Cut Line= 4
2183831.14877279671263.7013109052183847.40035796671279.952896066
2183850.30242673671349.0221329982183866.55401189671381.525303319
#Sta/Elev= 28
       0  1849.1     2.1 1848.29     4.6 1847.21     7.1 1845.97    10.3 1844.02
    13.4 1841.98    18.4 1839.71    28.7 1833.24    32.2 1831.13    36.2 1829.95
    44.2 1830.48    48.2 1829.84    52.2 1828.88    56.2 1828.52    64.2 1828.73
    68.41828.989    72.3 1829.75    76.3 1830.81    80.3 1832.09    84.3 1833.14
    88.3 1833.81    92.3  1834.1    96.8 1834.25    99.6 1834.43   105.7 1835.01
   110.2 1835.29   123.1 1835.77   128.5 1835.89
#Mann= 3 ,-1,0
       0     .08       0    52.2    .045       0    68.4      .1       0
Bank Sta=52.2,68.4
XS Rating Curve= 0 ,0
Exp/Cntr(USF)=0,0
Exp/Cntr=0.3,0.1

Type RM Length L Ch R = 1 ,5818    ,79.7,79,77.8
XS GIS Cut Line= 2
2183742.15617451671313.6991674222183851.23255933671390.132254596
#Sta/Elev= 28
       0 1858.52     2.5 1857.43    12.2 1852.23      13 1851.74    15.4 1850.08
    18.3 1847.87    33.9 1834.61    35.5 1833.61    41.5  1830.3    44.2 1829.52
    46.4 1829.09    51.3 1829.08    54.9 1828.73    55.6 1828.63    58.5  1828.5
      66 1828.43      70 1828.59    70.8 1828.75    72.9 1829.35    75.7 1830.62
    80.6 1832.44    82.7 1832.98    85.5 1833.35    95.3 1833.79   100.2 1833.78
   109.9 1834.45   117.6 1834.81   133.2 1835.96
#Mann= 4 ,-1,0
       0     .08       0      10      .1       0    54.9    .045       0
    70.8      .1       0
Bank Sta=54.9,70.8
XS Rating Curve= 0 ,0
Exp/Cntr(USF)=0,0
Exp/Cntr=0.3,0.1

Type RM Length L Ch R = 1 ,5739    ,89.1,89.7,90.1
XS GIS Cut Line= 2
2183689.60842708671378.9857627172183814.60837172671452.234137925
#Sta/Elev= 30
       0 1858.59       3 1857.03     9.3 1853.26    16.9  1849.4    21.5 1846.73
    26.9 1843.12    30.8 1840.34    35.4 1837.44    44.7 1832.51    47.3 1831.47
    50.2 1830.49    53.2 1829.86    58.6 1828.99    61.9 1828.14    63.2 1827.82
    64.9 1827.59    67.6 1827.33    70.7 1827.28    77.2 1827.32    81.8 1827.54
    84.61828.132    91.1 1829.83   100.3 1832.88     105 1833.34   109.6 1833.21
     123    1834   126.3 1834.56   132.8 1835.93   137.4 1836.57   144.9 1837.29
#Mann= 3 ,-1,0
       0      .1       0    61.9    .045       0    84.6      .1       0
Bank Sta=61.9,84.6
XS Rating Curve= 0 ,0
Exp/Cntr(USF)=0,0
Exp/Cntr=0.3,0.1

Type RM Length L Ch R = 1 ,5649    ,96.4,94.3,93.2
XS GIS Cut Line= 2
2183652.98423947671454.6226718992183771.61476019671534.240471039
#Sta/Elev= 30
       0 1855.57     3.8 1853.81     8.7 1851.34    15.7 1847.15    26.1  1841.5
    27.2 1840.86      33 1836.71    35.9 1834.77    38.7 1832.98    42.4 1830.94
    44.5 1830.04    47.4 1829.04      52 1828.73    56.8 1828.92    58.9 1828.77
    61.7  1828.4    64.7 1827.76    67.6 1827.37    76.1 1827.06    79.1 1827.17
    80.9 1827.42      82 1827.75    85.7 1829.17    90.6 1830.47   100.2 1831.21
     105  1832.5   109.8 1833.62   128.1  1835.6   138.7 1836.53   142.9 1836.77
#Mann= 3 ,-1,0
       0      .1       0    64.7    .045       0      82      .1       0
Bank Sta=64.7,82
XS Rating Curve= 0 ,0
Exp/Cntr(USF)=0,0
Exp/Cntr=0.3,0.1

Type RM Length L Ch R = 1 ,5555    ,73.2,72.9,72.5
XS GIS Cut Line= 2
2183593.40386461671534.4962279662183728.83374095671611.239824557
#Sta/Elev= 29
       0 1851.59     1.1  1851.3     3.2 1850.59     9.9 1847.49    12.4  1846.2
    15.7 1844.27    18.7 1842.83    21.6 1841.54    27.5 1839.22    30.8 1837.79
    44.6 1831.54      48 1830.43    53.8 1828.72    58.71827.133      63 1826.12
    67.6 1826.06    72.1 1825.85    77.4 1825.92    80.3 1826.08    81.3  1826.2
    85.1 1827.12    90.5 1828.41    94.7  1829.6   100.8 1831.87   104.3 1832.91
   108.9 1833.22   122.7 1833.64   136.5 1834.44   155.7    1835
#Mann= 3 ,-1,0
       0      .1       0    58.7    .045       0    85.1      .1       0
Bank Sta=58.7,85.1
XS Rating Curve= 0 ,0
Exp/Cntr(USF)=0,0
Exp/Cntr=0.3,0.1

Type RM Length L Ch R = 1 ,5482    ,70.7,71.2,71.7
XS GIS Cut Line= 2
2183559.22394344671601.5662619612183699.16814899671673.795529341
#Sta/Elev= 30
       0 1846.54     5.6  1844.7    10.1 1842.76    25.3 1835.41    28.1 1834.16
      36 1830.02    37.1 1829.53      39 1828.91    41.6 1828.24    46.1 1827.82
    51.5 1827.51    55.1 1827.18    60.11826.099    64.1 1825.51    68.7 1825.47
    73.1  1825.7    75.11826.115    80.6  1827.5    82.1 1827.77    89.5 1827.71
    91.1 1827.82    92.5  1828.1    95.4 1829.05   100.1 1831.16   101.4 1831.58
   104.6 1832.33   116.2  1833.1   131.1 1833.55     140 1833.98   157.5 1834.26
#Mann= 4 ,-1,0
       0      .1       0    60.1    .045       0    75.1      .1       0
  157.48     .05       0
Bank Sta=60.1,75.1
XS Rating Curve= 0 ,0
Exp/Cntr(USF)=0,0
Exp/Cntr=0.3,0.1

Type RM Length L Ch R = 1 ,5411    ,105.1,111.2,115.6
XS GIS Cut Line= 2
2183536.00739321671667.346487611 2183670.1474612671742.800275856
#Sta/Elev= 27
       0 1842.66     3.7    1841     9.4 1838.65    18.5  1834.3    27.7 1829.72
    30.8 1828.83    32.3  1828.5    42.6 1826.73    48.5 1825.41    51.4 1824.85
    54.3 1824.76    57.3 1824.99    59.9 1825.33    64.4 1826.29      69 1826.97
    77.2 1827.36    83.7 1827.03    87.4 1827.24    95.5 1828.09    98.4 1828.53
   104.3 1829.62   110.3 1830.96   114.9 1831.86   119.5 1832.34   124.1 1832.72
   133.6 1833.19   153.9 1833.59
#Mann= 3 ,-1,0
       0      .1       0    48.5    .045       0    59.9      .1       0
Bank Sta=48.5,59.9
XS Rating Curve= 0 ,0
Exp/Cntr(USF)=0,0
Exp/Cntr=0.3,0.1

Type RM Length L Ch R = 1 ,5299    ,88.7,88.4,88.1
XS GIS Cut Line= 3
2183491.04269301671731.6662432012183551.98613736671821.630375339
2183582.14721742671854.097009937
#Sta/Elev= 30
       0 1840.36     9.2 1838.03    16.3 1835.82      26 1832.62    30.8 1830.69
    35.6 1828.54    39.3 1827.43    42.2 1826.95    45.1 1826.73      48 1826.69
      55 1826.86    56.6 1826.72    59.1 1826.31    64.11824.749    66.2 1824.35
    68.2 1824.18      71 1824.11    74.3 1824.21    76.8 1824.75    85.4 1827.27
    88.3 1828.35    94.7 1831.14    98.5 1832.61    99.8 1833.04   103.3 1833.84
   108.5 1834.44   120.7 1835.33   132.4 1835.84   144.2 1836.08     153 1836.59
#Mann= 3 ,-1,0
       0      .1       0    64.1    .045       0    76.8      .1       0
Bank Sta=64.1,76.8
XS Rating Curve= 0 ,0
Exp/Cntr(USF)=0,0
Exp/Cntr=0.3,0.1

Type RM Length L Ch R = 1 ,5211    ,82.1,80.3,75.4
XS GIS Cut Line= 3
2183422.55386983671787.3859637512183488.72103798671883.154233446
 2183525.2871046 671917.97905879
#Sta/Elev= 30
       0 1835.02    11.1 1831.29    16.8  1829.9    21.6 1829.54    26.5 1829.48
    36.2 1829.98    41.1 1829.78    45.9 1829.07    55.7 1826.34    59.1 1825.83
    62.8 1825.64    65.4  1825.4    67.71824.939    70.2 1824.41    71.5 1824.35
    75.1 1824.66    77.2 1825.04      80 1825.95    84.8 1827.94    89.7 1829.41
    94.6 1830.54    99.4 1831.15   101.4 1831.32     114 1831.74   116.4 1831.94
   125.1 1832.75   134.4 1833.85   142.9 1834.68   157.1 1835.89   166.9 1836.95
#Mann= 4 ,-1,0
       0      .1       0    67.7    .045       0    77.2      .1       0
   156.4     .06       0
Bank Sta=67.7,77.2
XS Rating Curve= 0 ,0
Exp/Cntr(USF)=0,0
Exp/Cntr=0.3,0.1

Type RM Length L Ch R = 1 ,5131    ,72.9,73.3,74.8
XS GIS Cut Line= 3
 2183358.7083567671826.2736853852183426.61676612 671917.97905879
2183460.28076395671942.356436531
#Sta/Elev= 28
       0 1841.54     2.5  1840.6       6 1839.11     9.2 1837.64    13.6 1835.97
    23.1 1831.74    28.5 1829.65    33.5 1827.56    37.4 1825.65    40.3 1824.57
    43.4 1823.76      46 1823.72    58.4 1823.76      63 1824.29    64.61824.583
    68.3 1825.36    69.7 1825.53    73.3 1825.71    78.3 1825.76    83.1 1826.11
    88.9 1827.13    96.6 1828.28   100.4 1828.64   114.1 1829.63   131.8 1831.94
   135.8 1832.29   145.7 1832.64   155.7 1833.59
#Mann= 3 ,-1,0
       0      .1       0    40.3    .045       0    64.6      .1       0
Bank Sta=40.3,64.6
XS Rating Curve= 0 ,0
Exp/Cntr(USF)=0,0
Exp/Cntr=0.3,0.1

Type RM Length L Ch R = 1 ,5057    ,109.6,108.2,107.5
XS GIS Cut Line= 3
2183287.31125259671854.076319138 2183359.0655654671946.472283572
2183406.24648341671978.909164703
#Sta/Elev= 30
       0 1845.19       9 1843.85    14.1 1842.81    24.2 1839.82    29.3 1837.83
      34 1835.51    39.9 1832.28    44.4 1829.25    48.4  1826.8    49.5 1826.22
    51.3 1825.54      57 1823.92    59.6  1823.3    62.7 1822.69    64.7 1822.57
    65.5 1822.64    67.41823.234    71.2 1824.49    73.1 1824.85    79.9 1825.48
    95.1 1827.51   100.2  1827.8   105.2 1827.63   110.3 1827.62   112.3 1827.85
   132.9 1831.01   135.9 1831.32   142.9 1831.59     160 1831.75   174.2 1832.32
#Mann= 3 ,-1,0
       0      .1       0    59.6    .045       0    67.4      .1       0
Bank Sta=59.6,67.4
XS Rating Curve= 0 ,0
Exp/Cntr(USF)=0,0
Exp/Cntr=0.3,0.1

Type RM Length L Ch R = 1 ,4949    ,93.9,102.1,108.1
XS GIS Cut Line= 4
2183209.17260135671917.2309675022183214.67318251671938.810170526
2183294.22004856672028.511955647 2183317.4917381672075.055334719
#Sta/Elev= 30
       0 1834.13     4.1 1832.89     8.2 1831.38    12.3 1830.15    16.5 1829.06
    20.6 1828.16      25 1827.34    30.8 1826.64    39.2 1825.33    47.7 1823.83
    52.2 1822.87    54.7 1822.42    56.2 1822.28    60.7 1822.16    64.7 1822.43
    67.5 1822.95    70.3 1823.59    73.2 1824.04    78.9 1823.62    84.2 1823.55
    87.3 1823.66    94.9 1824.04   105.6 1824.89   121.7 1825.58   132.7 1826.43
   147.4 1826.92   151.9  1827.4   160.8 1829.92   164.4 1830.63   194.2 1834.15
#Mann= 3 ,-1,0
       0      .1       0    52.2    .045       0    67.5      .1       0
#XS Ineff= 2 , 0
                          108.53         1828.51
Permanent Ineff=
       F       F
Bank Sta=52.2,67.5
XS Rating Curve= 0 ,0
Exp/Cntr(USF)=0,0
Exp/Cntr=0.3,0.1

Type RM Length L Ch R = 1 ,4847    ,96.4,92.7,90.5
XS GIS Cut Line= 4
2183129.45465417 671919.916461292183145.70623933671953.000045367
 2183161.9578245672060.9570039322183174.72692712672080.110657871
#Sta/Elev= 30
       0 1840.26     5.9 1839.23    32.6 1833.26    41.1 1829.22    49.2 1824.82
    53.2 1823.54    57.3 1822.88    60.3 1822.74    69.4 1822.96    77.5 1822.62
    81.5 1822.79    85.6 1822.49    89.6 1821.37    92.1 1821.01    93.7 1820.78
   101.8 1820.61   105.8 1820.71   106.81820.926   109.9  1821.6   113.9 1823.61
   117.9 1824.73     122  1825.2   130.1 1824.66   134.1 1824.63   138.2 1825.11
   146.3 1827.28   151.1 1828.26   162.2 1829.38   165.5 1829.46   169.1 1829.25
#Mann= 3 ,-1,0
       0      .1       0    92.1    .045       0   106.8      .1       0
#XS Ineff= 2 , 0
                          122.16         1835.98
Permanent Ineff=
       F       F
Bank Sta=92.1,106.8
XS Rating Curve= 0 ,0
Exp/Cntr(USF)=0,0
Exp/Cntr=0.3,0.1

Type RM Length L Ch R = 1 ,4755    ,74.6,67.2,61.1
XS GIS Cut Line= 3
2183049.93796964671956.4825279012183076.05658865672044.705418772
2183095.21024259 672095.20141552
#Sta/Elev= 30
       0 1838.82     4.9 1837.12     8.8 1835.54    17.4 1831.51    25.8  1826.8
    29.9 1824.17    34.1 1821.19    36.91820.207    38.3 1819.75    50.8 1819.22
      55 1819.54      57 1820.24    59.1 1821.01    63.3 1822.27    66.7 1822.49
    71.6 1822.64    73.2 1822.79    75.8 1823.11      80 1823.87    84.2 1824.37
      92 1824.39   101.1 1824.09   105.3 1823.64   109.6 1822.92   113.9 1822.62
   118.2  1823.2   126.7 1825.74     131 1826.73   135.3  1827.2     146 1827.54
#Mann= 3 ,-1,0
       0      .1       0    36.9    .045       0      57      .1       0
#XS Ineff= 2 , 0
                           88.22         1834.71
Permanent Ineff=
       F       F
Bank Sta=36.9,57
XS Rating Curve= 0 ,0
Exp/Cntr(USF)=0,0
Exp/Cntr=0.3,0.1

Type RM Length L Ch R = 1 ,4687    ,65.8,68.4,72
XS GIS Cut Line= 3
2182970.72745488671998.548810888 2183060.7436198672096.285797931
2183092.27226826672104.167960046
#Sta/Elev= 30
       0 1826.22     3.6 1825.11     5.7 1824.68     8.5 1824.18    11.4 1823.91
    14.5 1823.74    19.8 1823.81    25.8 1824.17    30.8  1823.8    37.6 1822.55
    47.1 1821.21    52.5 1820.09    56.7 1819.34    59.5 1819.21    63.4 1819.37
    67.1 1820.11    70.8 1821.29      73 1821.81    74.3 1821.96    78.9 1821.96
      96 1821.18   101.5 1821.59   117.8 1825.31   123.2 1826.34   124.6 1826.47
   128.7 1826.69     132 1826.69   140.5 1826.98   152.9 1826.91   165.4  1827.3
#Mann= 3 ,-1,0
       0      .1       0    52.5    .045       0    67.1      .1       0
#XS Ineff= 2 , 0
            25.8 1826.28
Permanent Ineff=
       F       F
Bank Sta=52.5,67.1
XS Rating Curve= 0 ,0
Exp/Cntr(USF)=0,0
Exp/Cntr=0.3,0.1

Type RM Length L Ch R = 1 ,4619    ,54.8,58.4,62.3
XS GIS Cut Line= 3
2182920.60448983671995.9820470372182973.32327634672114.199802737
2182987.65448019672124.231645429
#Sta/Elev= 30
       0 1833.02     6.6 1828.89    10.1 1826.81    14.4 1824.57    18.8 1823.03
    23.2 1822.59    27.6 1822.76    36.3 1823.38    45.1  1823.6    53.9 1823.98
    62.6 1824.14      67 1824.02    71.4 1823.28    80.1 1821.26    84.5 1820.95
    88.9 1820.85    93.3 1820.54    94.5 1820.35    99.51819.128     102 1818.61
   106.4  1818.4   109.6 1819.11   110.8 1819.43   112.7 1820.27   116.8  1822.4
   119.6 1823.72   123.9 1825.19   134.6  1825.5   139.4 1825.28   146.9 1825.18
#Mann= 3 ,-1,0
       0      .1       0    99.5    .045       0   109.6      .1       0
#XS Ineff= 2 , 0
           61.19 1829.72
Permanent Ineff=
       F       F
Bank Sta=99.5,109.6
XS Rating Curve= 0 ,0
Exp/Cntr(USF)=0,0
Exp/Cntr=0.3,0.1
